--- CRKDFK.prj (project) ---

Proj Title=CRKDFK
Current Plan=p01
Default Exp/Contr=0,0
English Units
Geom File=g01
Flow File=f01
Plan File=p01
BEGIN DESCRIPTION:
----------MODEL BY WOOD PLC 2021----------
Stream Name: Crooked Fork
Flood Zone: Enhanced Approximate
Pocahontas County, WV
HEC-RAS Version: RAS 6.1.0
Vertical Datum: NAVD88
Projection: NAD 1983 StatePlane West Virginia S FIPS 4702 (US Feet)
Terrain: 1-meter LIDAR (FEMA Region III 3DEP collected 2016-2018)
Land Use: 2019 NLCD
Hydrologic Method:
WV SIR2010-5033 regression equations
Model Notes:
KWSEL used at tie in, Crooked Fork is more dominant in facc and flow than Old Field Fork upstream of their confluence
END DESCRIPTION:
DSS Export Rating Curves= 0
DSS Export Rating Curve Sorted= 0
DSS Export Volume Flow Curves= 0
DXF OffsetX= 0
DXF OffsetY= 0
DXF ScaleX= 0
DXF ScaleY= 0

--- CRKDFK.p01 (plan) ---

Plan Title=Floodplain
Program Version=6.10
Short Identifier=Floodplain
Geom File=g01
Flow File=f01
Subcritical Flow
K Sum by GR= 0
Std Step Tol= 0.01
Critical Tol= 0.01
Num of Std Step Trials= 20
Max Error Tol= 0.3
Flow Tol Ratio= 0.001
Split Flow NTrial= 30
Split Flow Tol= 0.02
Split Flow Ratio= 0.02
Log Output Level= 0
Friction Slope Method= 1
Unsteady Friction Slope Method= 2
Unsteady Bridges Friction Slope Method= 1
Parabolic Critical Depth
Global Vel Dist= 0 , 0 , 0
Global Log Level= 0
CheckData=True
Encroach Param=-1 ,0,0, 0
Mapping Interval=1HOUR
Computation Time Step Use Courant=        0
Computation Time Step Use Time Series=    0
Computation Time Step Count To Double=0
Computation Time Step Max Doubling=0
Computation Time Step Max Halving=0
Computation Time Step Residence Courant=0
Run HTab= 0
Run UNet= 0
Run Sediment= 0
Run PostProcess= 0
Run WQNet= 0
Run RASMapper=-1
UNET Theta= 0
UNET Theta Warmup= 0
UNET ZTol= 0
UNET ZSATol= 0
UNET MxIter= 0
UNET Max Iter WO Improvement= 0
UNET MaxInSteps= 0
UNET DtIC= 0
UNET DtMin= 0
UNET MaxCRTS= 0
UNET WFStab= 0
UNET SFStab= 0
UNET WFX= 1
UNET SFX= 1
UNET Gravity=32.174
UNET 1D Methodology=Finite Difference
UNET DSS MLevel= 1
UNET Pardiso=0
UNET DZMax Abort= 0
UNET Use Existing IB Tables= 0
UNET Froude Reduction=False
UNET Froude Limit= 0
UNET Froude Power= 0
UNET D1 Cores= 0
UNET WindReference=Eulerian
UNET WindDragFormulation=Hsu (1988)
UNET D2 Coriolis=0
UNET D2 Cores= 0
UNET D2 Theta= 1
UNET D2 Theta Warmup= 1
UNET D2 Z Tol= 0.01
UNET D2 Volume Tol= 0.01
UNET D2 Max Iterations= 20
UNET D2 Equation= 0
UNET D2 RampUpFraction=0.1
UNET D2 TimeSlices= 1
UNET D2 Turbulence Formulation=Non-Conservative (original)
UNET D2 Eddy Viscosity=0.3
UNET D2 Transverse Eddy Viscosity=0.1
UNET D2 Smagorinsky Mixing=0
UNET D2 BCVolumeCheck=0
UNET D2 Cores=0
UNET D2 SolverType=PARDISO (Direct)
UNET D2 Minimum Iterations= 2147483647
UNET D2 Maximum Iterations= 2147483647
UNET D2 Restart Number= 10
UNET D2 Relaxation Coeff=1.3
UNET D2 SOR Precondition Iterations= 10
UNET D2 ILUT Maximum Fill= 8
UNET D2 ILUT Tolerance=1E-08
UNET D1D2 MaxIter= 0
UNET D1D2 ZTol=0.01
UNET D1D2 QTol=0.1
UNET D1D2 MinQTol=1
Write IC File= 0
Write IC File at Fixed DateTime=0
Write IC File at Sim End=0
Echo Input=False
Echo Parameters=False
Echo Output=False
Write Detailed= 0
HDF Write Warmup=0
HDF Write Time Slices=0
HDF Flush=0
HDF Compression= 1
HDF Chunk Size= 1
HDF Spatial Parts= 1
HDF Use Max Rows=0
HDF Fixed Rows= 1
Calibration Method= 0
Calibration Iterations= 20
Calibration Max Change=0.05
Calibration Tolerance=0.2
Calibration Maximum=1.5
Calibration Minimum=0.5
Calibration Optimization Method= 1
WQ AD Non Conservative
WQ ULTIMATE=-1
WQ Max Comp Step=1HOUR
WQ Output Interval=15MIN
WQ Output Selected Increments= 0
WQ Output face flow=0
WQ Output face velocity=0
WQ Output face area=0
WQ Output face dispersion=0
WQ Output cell volume=0
WQ Output cell surface area=0
WQ Output cell continuity=0
WQ Output cumulative cell continuity=0
WQ Output face conc=0
WQ Output face dconc_dx=0
WQ Output face courant=0
WQ Output face peclet=0
WQ Output face adv mass=0
WQ Output face disp mass=0
WQ Output cell mass=0
WQ Output cell source sink temp=0
WQ Output nsm pathways=0
WQ Output nsm derived pathways=0
WQ Create Restart=0
WQ Fixed Restart=0
WQ System Summary=0
WQ Write To DSS=0
Sorting and Armoring Iterations= 10
XS Update Threshold= 0.02
Bed Roughness Predictor= 0
Hydraulics Update Threshold= 0.02
Energy Slope Method= 1
Volume Change Method= 1
Sediment Retention Method= 0
Sediment TS Multiplier= 1
Warm Up Method= 0
XS Weighting Method= 0
Number of US Weighted Cross Sections= 1
Number of DS Weighted Cross Sections= 1
Upstream XS Weight=0
Main XS Weight=1
Downstream XS Weight=0
Number of DS XS's Weighted with US Boundary= 1
Upstream Boundary Weight= 1
Weight of XSs Associated with US Boundary= 0
Number of US XS's Weighted with DS Boundary= 1
Downstream Boundary Weight= 0.5
Weight of XSs Associated with DS Boundary= 0.5
Percentile Method= 0
Sediment Output Level= 3
Mass or Volume Output= 0
Output Increment Type= 1
Profile and TS Output Increment= 1
Transport Output Increment 1
XS Output Flag= 0
XS Output Increment= 10
Read HDF5 Sediment Hotstart= 0
Sediment Hotstart Type= 0
Write Gradation File= 0
Read Gradation Hotstart= 0
Write HDF5 File= 1
Write Binary Output= 1
Write DSS Sediment File= 0
DSS Sediment Output Type= 1
SV Curve= 0
Specific Gage Flag= 0
Subcell Erosion Methods= 0
Subcell Deposition Methods= 0
Advection Scheme= 1
Matrix Solver= 0
Implicit Weighting Factor= 1
Maximum Outer Loop Convergence Iterations= 5
Convergence Maximum Absolute= 0.001
Convergence RMSE= 0.0001
Grain Fractions Max Abs Error= 0.001
Max Subgrid Regions= 1
Max Subgrid Length Scale= 3.402823E+38
Initial Layer Thickness= 3.402823E+38
Min Layer Thickness= 3.402823E+38
Max Layer Thickness= 3.402823E+38
Number of Layers= 5

--- CRKDFK.f01 (steady flow) ---

Flow Title=Flow
Program Version=6.10
Number of Profiles= 6
Profile Names=01pct,10pct,04pct,02pct,0_2pct,01plus
River Rch & RM=CRKDFK,Main            ,10897
     671     357     473     569     934     992
River Rch & RM=CRKDFK,Main            ,8991
     777     415     549     659    1080    1150
River Rch & RM=CRKDFK,Main            ,7792
     887     477     629     754    1230    1310
River Rch & RM=CRKDFK,Main            ,6471
     987     533     701     840    1370    1460
River Rch & RM=CRKDFK,Main            ,1703
    1120     605     794     950    1540    1650
River Rch & RM=CRKDFK,Main            ,0
    2030    1100    1430    1720    2860    2930
Boundary for River Rch & Prof#=CRKDFK,Main            , 1
Up Type= 0
Dn Type= 1
Dn Known WS=3049.3
Boundary for River Rch & Prof#=CRKDFK,Main            , 2
Up Type= 0
Dn Type= 1
Dn Known WS=3048
Boundary for River Rch & Prof#=CRKDFK,Main            , 3
Up Type= 0
Dn Type= 1
Dn Known WS=3048.4
Boundary for River Rch & Prof#=CRKDFK,Main            , 4
Up Type= 0
Dn Type= 1
Dn Known WS=3048.9
Boundary for River Rch & Prof#=CRKDFK,Main            , 5
Up Type= 0
Dn Type= 1
Dn Known WS=3050.7
Boundary for River Rch & Prof#=CRKDFK,Main            , 6
Up Type= 0
Dn Type= 1
Dn Known WS=3050.9
DSS Import GetInterval= 0
DSS Import GetPeak= 0
DSS Import FillOption= 0

--- CRKDFK.g01 (geometry) ---

Geom Title=Geometry
Program Version=6.10

River Reach=CRKDFK          ,Main
Reach XY= 30
2219042.77704822486320.304980561 2219379.6979623486173.868921727
 2219570.0401013486418.6171198932219761.61714597486459.590135068
2219909.19001356486643.5769718142220270.16895039486631.271878317
2220861.74388272486884.6378413892221404.10303421486554.411139637
2221580.55707763486345.7799952332221928.32114589486139.883097306
2222212.61093163485865.3019535542222364.79993172485825.820077151
2222409.35200797485668.128135309 2222731.4018888485379.789145067
2223153.96502006 485181.824974062223257.34998389485042.618887648
2223518.29500005485062.7080863122223645.31311873 485163.80696547
2224595.03005131485097.2729778142224881.51897964 484995.00710623
2224939.57004464484787.8461032212225183.50295572484793.000948563
2225606.63399921484591.8589623872225956.05685681484524.891904727
2225911.97098698484195.1100839822226084.76788548484013.927047387
2226143.75005098483639.3510248962226364.95498914483444.454104975
2226998.17911638483666.770917565 2227178.4166168 484173.32305406

Type RM Length L Ch R = 1 ,10897   ,251.4,251.4,251.4
XS GIS Cut Line= 4
2218983.03192183 486616.63284336  2219077.795037486430.226598186
2218997.62435462486145.4130150142218921.54158634486051.426646124
#Sta/Elev= 30
       0 3345.66    12.8 3338.04    48.7 3312.29    57.7 3307.17    83.7 3286.55
    93.6 3281.61   102.6  3278.8   120.5 3277.95     134  3280.4   152.2 3280.91
   169.9 3279.23   184.9 3275.48   196.7 3277.06   211.3 3276.55   226.8  3278.9
   251.8 3278.66   272.9 3281.21     285 3281.34   293.3 3280.21   305.3 3275.86
     315 3275.14   322.4 3273.27  333.47  3275.1     339 3278.73   343.2 3279.43
   401.3 3279.28   422.1 3278.19     435 3281.26     531 3287.85   625.9 3297.63
#Mann= 3 ,-1,0
       0      .1       0     315    .045       0  333.47      .1       0
#XS Ineff= 2 , 0
          281.97 3286.18
Permanent Ineff=
       F       F
Bank Sta=315,333.47
XS Rating Curve= 0 ,0
Exp/Cntr=0.3,0.1

Type RM Length L Ch R = 1 ,10645   ,210.7,226.4,245.2
XS GIS Cut Line= 5
2219132.93119526 486697.053583012219311.21470202486342.800610427
2219276.86950975486241.2165156562219244.73098837 486155.51379198
2219232.37001861486048.385387384
#Sta/Elev= 30
       0 3341.74     8.8 3338.03    22.2 3330.62      53 3312.36    84.9 3291.12
    98.4 3284.21   107.3  3278.3   116.3 3273.96   122.9 3272.03   161.1 3269.68
   192.4 3272.17   210.8 3267.26   214.8 3267.18   225.7 3269.43   246.1 3268.03
   259.6 3269.14     273 3268.37   285.3 3265.73   303.2 3268.79   327.5 3266.94
     376 3269.22   395.5 3266.89   419.4 3267.39   436.3 3264.08   499.6 3268.21
   549.6 3269.86   580.9 3269.93   621.9 3298.71   662.1  3305.3   703.2 3315.16
#Mann= 3 ,-1,0
       0      .1       0   549.6    .045       0   580.9      .1       0
#XS Ineff= 2 , 0
             509 3276.97
Permanent Ineff=
       F       F
Bank Sta=549.6,580.9
XS Rating Curve= 0 ,0
Exp/Cntr(USF)=0,0
Exp/Cntr=0.3,0.1

Type RM Length L Ch R = 1 ,10419   ,220.8,218.3,218.5
XS GIS Cut Line= 3
2219205.95809048486697.4072557272219390.59043155486326.095174681
2219494.16955366486151.539799117
#Sta/Elev= 30
       0  3315.6    22.9  3301.3    31.7 3298.22    44.9 3289.07    58.3 3282.39
    79.4 3275.34   103.8 3270.57   138.7 3271.14     170 3265.72   187.9 3267.79
   210.2 3263.92   223.6 3263.75   259.4 3267.03   279.9 3262.93   299.6 3264.87
   356.9 3263.54   383.7 3259.98   402.3  3263.7   436.9 3262.37   457.6 3259.67
   480.5 3262.29   490.2  3259.6   495.3 3258.03   511.8 3259.67   527.2 3260.92
     532 3262.05   558.9 3276.28   573.9 3286.62   587.8 3298.85   617.7 3316.41
#Mann= 4 ,-1,0
       0      .1       0   490.2    .045       0   511.8      .1       0
   527.2     .06       0
Bank Sta=490.2,511.8
XS Rating Curve= 0 ,0
Exp/Cntr(USF)=0,0
Exp/Cntr=0.3,0.1

Type RM Length L Ch R = 1 ,10201   ,209.6,213,208.7
XS GIS Cut Line= 3
2219354.45692073 486767.464028262219623.88876392 486333.00746702
2219674.62744261486218.280124752
#Sta/Elev= 30
       0 3308.01    52.3 3277.79    73.3 3269.07    94.3 3263.17   143.9 3261.26
   162.6 3258.78   219.2 3259.99   233.3 3257.07   247.4 3260.03   285.1 3258.62
   334.1 3259.13   339.9 3258.08   346.3 3254.07   352.4 3252.74   374.5 3253.86
   383.9 3256.11   393.3 3253.84  422.47 3253.83   427.1 3255.13   440.4 3254.73
   456.1 3258.11   487.5 3261.24   501.6 3270.17   511.9 3278.98   521.8 3283.78
   531.7 3289.68   541.6 3293.72   593.2 3308.58   623.5 3320.09   636.7 3327.32
#Mann= 5 ,-1,0
       0      .1       0   393.3    .045       0  422.47      .1       0
   521.8     .06       0   623.5      .1       0
Bank Sta=393.3,422.47
XS Rating Curve= 0 ,0
Exp/Cntr=0.3,0.1

Type RM Length L Ch R = 1 ,9988    ,165.2,171.7,167.2
XS GIS Cut Line= 3
2219616.19180955486964.9473756452219637.40277767486652.364687468
2219852.86155917486340.898366035
#Sta/Elev= 30
       0 3268.27    55.9 3260.76      80 3255.17   112.4 3252.06   136.1 3252.78
   164.1 3251.01   200.2 3251.69   240.3 3248.44   252.3 3249.96   288.4 3249.45
   296.4 3251.72   308.5 3252.67   353.3 3252.97   360.7 3253.12   385.3 3249.96
   419.3 3249.89     429 3245.89   449.8 3245.07   472.8 3249.84   511.7 3249.51
  523.21  3247.8   543.2  3247.8   560.4 3254.04   578.3 3266.75   604.1 3274.03
   618.7 3276.72   642.5 3284.95   662.5 3293.93   672.2  3296.4     692    3304
#Mann= 6 ,-1,0
       0      .1       0     280     .12       0   353.3      .1       0
  523.21    .045       0   543.2      .1       0   663.3     .06       0
#XS Ineff= 2 , 0
          351.93 3255.87
Permanent Ineff=
       F       F
Bank Sta=523.21,543.2
XS Rating Curve= 0 ,0
Exp/Cntr(USF)=0,0
Exp/Cntr=0.3,0.1

Type RM Length L Ch R = 1 ,9816    ,155.8,148.7,141.3
XS GIS Cut Line= 4
2219727.13112905486923.4429890922219805.56936554486662.590596246
2219890.05840492 486539.516011322219935.53902323 486387.58221065
#Sta/Elev= 30
       0 3269.89    27.4 3264.78      38 3260.01    48.3 3253.84    63.7 3247.05
    98.4 3243.74   119.3  3242.9     136 3245.11   161.1 3245.48   194.5 3243.92
   261.3    3248   288.7 3248.44   301.2 3247.96   312.9 3245.44   332.3 3245.68
   341.4 3243.23   351.7 3242.11   358.7 3243.23   366.3 3244.68   400.3 3244.35
   410.5 3243.25   436.6 3245.58   483.1 3245.06   490.9 3246.08   508.8 3256.82
   528.5 3271.17   536.8 3275.77   547.4 3279.84   568.5 3292.39   580.3 3297.77
#Mann= 8 ,-1,0
       0      .1       0      30     .12       0     210      .1       0
  322.39     .12       0   341.4    .045       0   358.7     .12       0
  441.67      .1       0  541.67     .06       0
#XS Ineff= 2 , 0
          298.82 3253.57  436.73         3251.91
Permanent Ineff=
       F       F
Bank Sta=341.4,358.7
XS Rating Curve= 0 ,0
Exp/Cntr=0.3,0.1

Type RM Length L Ch R = 1 ,9667    ,206.4,211.6,216.6
XS GIS Cut Line= 3
 2219984.5928349487006.2529451542219981.24373467486579.800849141
2220044.87663904486427.974972027
#Sta/Elev= 30
       0 3292.55    13.1  3288.4    29.1 3281.03    45.1 3275.13    93.1 3261.88
   101.1 3257.76   121.6 3244.07   133.1 3238.04   141.1 3236.04   157.1 3234.48
   165.1  3234.6   185.1 3238.34   202.3 3237.71   222.4 3239.16   245.1 3236.98
   313.1 3239.47   337.1 3242.41   353.1 3239.78   365.1 3239.65   389.1 3239.59
   393.1 3240.99   413.1 3239.85   427.7 3242.04     438  3240.1   459.7 3240.82
     503 3238.97   507.4 3241.15   524.7  3257.6   537.5  3267.2   591.1 3293.82
#Mann= 5 ,-1,0
       0      .1       0     190     .12       0   353.1    .045       0
   365.1     .12       0  591.09     .06       0
#XS Ineff= 2 , 0
          335.72 3247.32  427.07          3247.2
Permanent Ineff=
       F       F
Bank Sta=353.1,365.1
XS Rating Curve= 0 ,0
Exp/Cntr(USF)=0,0
Exp/Cntr=0.3,0.1

Type RM Length L Ch R = 1 ,9456    ,297.2,297.2,294.8
XS GIS Cut Line= 3
2220062.78539287487056.1236081692220185.13459365486590.499115458
2220183.43325615486452.101938729
#Sta/Elev= 30
       0 3306.28    15.5 3301.63    27.9 3296.55    40.3  3289.8    52.7 3286.35
    60.9 3281.44    73.4  3276.1   118.8 3260.57   170.5 3248.15   222.2 3234.16
   234.6 3231.78   241.6 3231.98     259 3230.61   292.5 3233.21   304.5 3232.85
   331.1 3235.72   363.8 3234.17   387.7 3234.83   408.4 3232.18   420.8 3234.61
   441.4 3235.14  444.373234.071   453.8 3232.58   465.3 3234.15   481.4 3243.94
   526.8 3249.82   554.7  3260.7   566.8 3265.36     583 3275.57   619.8 3292.91
#Mann= 6 ,-1,0
       0     .12       0    40.3      .1       0   241.6     .12       0
  444.37    .045       0   465.3     .12       0   554.7     .06       0
#XS Ineff= 1 ,-1
  184.86     380 3237.45
Permanent Ineff=
       F
Bank Sta=444.37,465.3
XS Rating Curve= 0 ,0
Exp/Cntr=0.3,0.1

Type RM Length L Ch R = 1 ,9159    ,165.8,167.4,168.3
XS GIS Cut Line= 3
2220366.52319004487163.9574730122220466.79390482 486622.04495831
2220519.74585532486484.595214456
#Sta/Elev= 30
       0 3308.53    23.2  3297.9    63.8 3276.07    79.3 3268.59   124.9 3251.89
   177.7  3230.5   206.2 3226.25   288.7 3224.56   309.3 3223.09   336.4 3224.97
     373 3225.97   413.7  3225.8   421.8 3224.95     434 3225.48   443.2 3223.76
   450.3  3222.6   458.4  3222.7   463.8 3223.79   470.6 3226.67   474.7 3227.05
   482.8 3223.72   486.9 3223.45   519.4 3226.06   535.7 3237.14   549.6 3241.22
   565.2  3244.2   590.6 3246.39     644 3255.56   680.6 3259.15   698.4 3261.92
#Mann= 7 ,-1,0
       0      .1       0      50     .12       0     310      .1       0
     350     .12       0   443.2    .045       0   463.8     .12       0
     550      .1       0
#XS Ineff= 2 , 0
          374.51 3229.25  475.15         3229.61
Permanent Ineff=
       F       F
Bank Sta=443.2,463.8
XS Rating Curve= 0 ,0
Exp/Cntr(USF)=0,0
Exp/Cntr=0.3,0.1

Type RM Length L Ch R = 1 ,8991    ,175.3,179.2,184.2
XS GIS Cut Line= 3
2220500.29713749487150.183274664 2220631.2743234486671.129731672
2220572.06545854486520.416257473
#Sta/Elev= 30
       0 3273.95     9.3 3268.72    33.3 3258.24    54.9 3250.79   108.2 3236.32
   137.5 3223.44     144 3221.81   212.5 3221.68   233.3 3218.08   241.7 3219.48
   266.4 3220.19   274.7 3219.58   290.5 3221.14     318 3221.72   336.9  3220.1
   349.4 3220.69   382.5 3217.62     411 3219.19     4213218.402   442.33218.262
   448.9 3220.51   469.6  3222.4   482.7 3228.71   489.2 3230.65   498.7 3231.64
   511.6 3230.71     527 3231.71   540.6  3235.5   556.1 3241.29   658.6 3255.26
#Mann= 8 ,-1,0
       0     .12       0      40      .1       0     240     .12       0
     421    .045       0   442.3     .12       0     460      .1       0
  536.64     .12       0  656.64      .1       0
#XS Ineff= 2 , 0
           346.5 3222.05
Permanent Ineff=
       F       F
Bank Sta=421,442.3
XS Rating Curve= 0 ,0
Exp/Cntr(USF)=0,0
Exp/Cntr=0.3,0.1

Type RM Length L Ch R = 1 ,8812    ,182,163.8,142
XS GIS Cut Line= 3
2220542.27860022487185.3635806612220817.17808792486744.848417982
2220830.69773486486546.560262915
#Sta/Elev= 30
       0  3280.5    18.7 3273.23    33.4 3263.78    56.8 3252.28   118.1 3234.33
   135.1 3227.29   146.4 3220.28   151.1  3218.9   215.1 3217.63   250.1 3219.06
   316.1 3214.55   326.7 3216.46     347 3215.79   353.8 3214.04   372.7 3214.97
   381.8 3213.18   393.4 3213.07     401 3212.06   415.1 3213.07   428.3 3214.56
     437 3217.89   457.6 3219.65   476.4 3219.54   500.9 3222.14   517.4 3229.38
   526.9 3232.03     551 3235.49   587.1 3239.22   707.4 3247.88     718 3249.65
#Mann= 5 ,-1,0
       0      .1       0   393.4    .045       0   415.1      .1       0
  519.25     .12       0  539.25      .1       0
#XS Ineff= 2 , 0
          371.34 3217.53
Permanent Ineff=
       F       F
Bank Sta=393.4,415.1
XS Rating Curve= 0 ,0
Exp/Cntr(USF)=0,0
Exp/Cntr=0.3,0.1

Type RM Length L Ch R = 1 ,8648    ,174.5,174.6,173.9
XS GIS Cut Line= 4
2220966.99556917487204.9662254942220992.67200427487034.162113741
2220884.38443015486830.9833664262220881.03532992486576.451748911
#Sta/Elev= 30
       0 3232.66    11.9 3229.25    48.3  3223.5   121.1 3217.88   125.2 3217.12
   137.3 3211.82   141.4 3210.92   232.8 3210.87   237.3 3210.46   246.4  3206.8
   250.7 3206.23   267.3 3209.39   274.3 3209.83   300.8 3209.93   318.9 3208.15
   332.5 3209.42   350.23207.106   359.7 3206.25   382.3 3207.04   391.4 3214.18
   394.9 3214.91   416.8    3214   428.6 3216.01   444.8 3217.14   468.1 3217.07
   472.8 3218.58   488.8 3228.32   503.7 3231.45   620.8 3242.28   657.5 3246.51
#Mann= 6 ,-1,0
       0     .12       0  342.72      .1       0   350.2    .045       0
   382.3      .1       0  412.96     .12       0  512.96      .1       0
#XS Ineff= 2 , 0
          276.06 3212.63
Permanent Ineff=
       F       F
Bank Sta=350.2,382.3
XS Rating Curve= 0 ,0
Exp/Cntr(USF)=0,0
Exp/Cntr=0.3,0.1

Type RM Length L Ch R = 1 ,8474    ,173.8,172.2,170.9
XS GIS Cut Line= 3
2221262.07745206487160.1962346822221012.08633126486703.162839928
2221006.08415611486556.095742813
#Sta/Elev= 30
       0  3215.6    30.8 3215.29   120.7 3209.47   170.7  3210.4   249.6 3206.41
   299.8 3206.41   304.4 3205.83   313.1 3202.52     318 3202.22   324.9 3202.86
   331.7 3206.31   333.7 3206.31     391 3204.75   427.5 3201.84   445.6 3200.53
   454.1 3202.02   459.4 3205.78   463.4 3206.88   478.1 3205.39     484 3205.99
     487 3207.27   504.6 3221.74   513.5 3226.01   538.9 3229.91     563 3235.38
     591 3244.06     619 3254.44     635 3263.11     651 3269.69   668.1 3279.15
#Mann= 8 ,-1,0
       0     .12       0     110      .1       0     160     .12       0
     280      .1       0     390     .12       0   427.5    .045       0
   454.1     .12       0     500      .1       0
#XS Ineff= 2 , 0
          333.63 3211.06
Permanent Ineff=
       F       F
Bank Sta=427.5,454.1
XS Rating Curve= 0 ,0
Exp/Cntr=0.3,0.1

Type RM Length L Ch R = 1 ,8301    ,198.7,200,200.9
XS GIS Cut Line= 2
2221431.49110308487047.9134171712221092.38578613486520.416257473
#Sta/Elev= 30
       0 3214.52    13.5 3212.58    93.6 3205.59   117.1 3204.75   131.6 3202.65
   164.9 3203.59   183.9 3201.34   282.2 3203.17   293.3  3201.1     302 3200.94
   328.6 3202.25   357.5 3202.02   374.9 3200.34   415.4 3200.02   433.8 3197.29
   442.6  3196.1     453 3197.35   464.5 3200.15   484.9 3200.77   488.3 3203.15
   496.4 3212.95   501.7  3217.7   526.3  3234.1   539.9 3238.16   554.3 3246.56
   564.4 3248.89   578.6  3256.7   597.7 3264.18     618 3275.25   627.1 3278.35
#Mann= 7 ,-1,0
       0      .1       0      40     .12       0      50      .1       0
     150     .12       0     270      .1       0   433.8    .045       0
     453      .1       0
#XS Ineff= 2 , 0
          328.15 3202.93
Permanent Ineff=
       F       F
Bank Sta=433.8,453
XS Rating Curve= 0 ,0
Exp/Cntr(USF)=0,0
Exp/Cntr=0.3,0.1

Type RM Length L Ch R = 1 ,8101    ,136.6,134.2,132.6
XS GIS Cut Line= 3
2221651.35019482486974.7859614372221519.98645573486860.422235638
2221243.34987575486351.967292555
#Sta/Elev= 30
       0  3242.2    57.3 3228.53   166.9  3209.7   197.1 3197.68   214.3 3196.47
   232.5 3199.15   246.2 3196.77   305.4 3197.27     315  3195.9   329.8  3197.2
   366.3 3194.93   405.5 3197.05   441.8 3194.45   473.9 3196.72   484.63192.896
   492.4 3191.19   502.3  3192.9   505.7 3194.91   512.6 3195.27   567.2 3193.19
   583.4 3194.83   604.1 3191.17   625.7 3194.66   646.9 3209.12   660.1 3225.62
   668.9 3232.39   707.3 3251.01   715.2 3256.33   724.3 3258.54     753 3272.26
#Mann= 9 ,-1,0
       0      .1       0      80     .12       0  214.17      .1       0
  334.17     .12       0  414.17      .1       0  444.17     .12       0
   484.6    .045       0   502.3     .12       0  624.17      .1       0
#XS Ineff= 2 , 0
           450.7 3199.85
Permanent Ineff=
       F       F
Bank Sta=484.6,502.3
XS Rating Curve= 0 ,0
Exp/Cntr(USF)=0,0
Exp/Cntr=0.3,0.1

Type RM Length L Ch R = 1 ,7967    ,178.9,175.5,174.8
XS GIS Cut Line= 3
2221761.84869053486780.7468629692221615.60464713486684.739323029
2221338.74569475486320.803764652
#Sta/Elev= 30
       0 3241.88    15.3 3237.27    28.4 3234.88    47.1 3228.97    79.4 3221.36
   115.8 3213.73   126.4 3213.16   159.9 3206.02   174.3 3200.85   185.6 3195.11
   191.3  3193.8   234.2 3192.27   246.7 3193.68   262.7 3191.39   282.7 3192.64
   390.5 3191.59   398.6 3189.31   418.4 3188.94   422.6 3189.37   460.9 3192.08
   510.9 3191.13   531.2 3188.95   536.3  3189.5   545.3 3197.26   556.7 3209.48
   571.4 3221.28   583.6 3226.82   606.6 3240.36   616.7 3243.84   632.2 3252.73
#Mann= 9 ,-1,0
       0      .1       0      80     .12       0  194.94      .1       0
  254.94     .12       0  364.94      .1       0  374.94     .12       0
   398.6    .045       0   422.6     .12       0  524.94      .1       0
#XS Ineff= 2 , 0
          363.74 3193.25
Permanent Ineff=
       F       F
Bank Sta=398.6,422.6
XS Rating Curve= 0 ,0
Exp/Cntr(USF)=0,0
Exp/Cntr=0.3,0.1

Type RM Length L Ch R = 1 ,7792    ,203.4,208.1,214.3
XS GIS Cut Line= 2
2221866.16854463486651.7857088412221394.80453965486171.148969331
#Sta/Elev= 30
       0 3245.78    65.7 3223.14    82.1 3219.72   110.1  3210.1     140  3202.9
   170.1 3188.88   231.4 3188.76   249.3 3186.86   283.3 3189.02   356.6 3184.56
   373.4 3184.92     397 3187.65   410.6 3185.35   424.7 3184.26     435 3185.28
   442.7 3188.03     470 3187.67   482.7 3185.56   489.8 3187.05   498.3 3193.24
   511.3 3206.71   528.4  3218.3   547.1 3226.42   575.1  3244.7   585.5 3249.57
   600.1  3259.2   608.7 3266.48   631.1 3279.97   659.1 3294.74   673.2  3299.8
#Mann= 4 ,-1,0
       0      .1       0   410.6    .045       0     435      .1       0
     590     .06       0
#XS Ineff= 2 , 0
          282.76 3190.82
Permanent Ineff=
       F       F
Bank Sta=410.6,435
XS Rating Curve= 0 ,0
Exp/Cntr(USF)=0,0
Exp/Cntr=0.3,0.1

Type RM Length L Ch R = 1 ,7584    ,228.3,223.7,219.1
XS GIS Cut Line= 4
2221984.00567248486483.7933092012221780.82692517486309.640097217
2221719.42675428 486185.723388692221541.92444206486036.130245062
#Sta/Elev= 30
       0 3241.97    89.7  3215.4   171.9 3198.84   194.6 3185.99   203.1 3183.39
   243.7 3181.02   248.5 3181.36     256 3184.13   272.6 3185.29     286 3181.88
   326.2 3183.14   331.1  3182.8   337.1 3180.35     346 3179.33   361.9 3180.26
   370.8 3182.64   388.6 3183.46   442.7 3182.62   468.2 3180.29   482.4 3182.76
   499.1 3190.55   513.6  3202.2   524.7 3206.47   536.3 3214.65   551.4 3221.74
   577.5 3239.89     593 3248.44   603.7 3257.14   614.2 3261.65     638 3276.15
#Mann= 4 ,-1,0
       0      .1       0   337.1    .045       0   361.9      .1       0
   565.9     .06       0
#XS Ineff= 2 , 0
           272.7 3187.22
Permanent Ineff=
       F       F
Bank Sta=337.1,361.9
XS Rating Curve= 0 ,0
Exp/Cntr(USF)=0,0
Exp/Cntr=0.3,0.1

Type RM Length L Ch R = 1 ,7360    ,177,177,177.8
XS GIS Cut Line= 3
2222117.68342916486329.4929289572221804.35031447485976.421544321
2221673.18338056485845.890787703
#Sta/Elev= 30
       0 3238.13     8.3 3236.49    38.1  3226.7    80.6 3216.31   160.9  3193.3
   185.5 3189.24   207.2 3187.23   219.7 3181.99     225 3180.84   247.8 3179.74
  254.933174.804   267.4 3173.82   279.5 3174.73   310.6  3177.8   341.3 3178.38
   363.8 3177.09   386.6 3178.25   446.1 3175.43   460.3 3177.38   474.5 3176.55
   488.6 3177.47   502.8 3176.37   510.7 3177.24   517.4 3181.25   536.7 3197.68
   550.8 3207.97   567.4 3217.77   624.1 3257.98   644.2 3272.21   657.1  3283.4
#Mann= 4 ,-1,0
       0      .1       0  254.93    .045       0   279.5      .1       0
   624.1     .07       0
#XS Ineff= 1 ,-1
   349.8   385.5    3180
Permanent Ineff=
       F
Bank Sta=254.93,279.5
XS Rating Curve= 0 ,0
Exp/Cntr=0.3,0.1

Type RM Length L Ch R = 1 ,7183    ,196,195.8,195.4
XS GIS Cut Line= 2
2222241.88639023486204.7016233292221808.73609376485713.500256194
#Sta/Elev= 30
       0 3224.17    20.7 3217.44   125.6 3190.82   143.4 3183.06     154 3176.13
   159.8 3173.67   196.7 3174.69   213.4 3173.31   247.4 3174.39   255.9 3172.09
   287.3 3171.91   292.8 3173.99   315.4 3174.93   377.8 3175.59   407.8 3174.39
     426 3175.75   468.3 3172.55   498.5 3173.88   516.7 3170.34     528 3171.57
   530.8 3173.13   533.7 3176.07     545 3191.61   556.3 3203.96     586    3222
     602  3235.8   621.5 3249.68     634 3259.38   644.7 3265.94   654.9 3274.38
#Mann= 4 ,-1,0
       0      .1       0   255.9    .045       0   287.3      .1       0
   621.5     .06       0
#XS Ineff= 2 , 0
           247.4    3176
Permanent Ineff=
       F       F
Bank Sta=255.9,287.3
XS Rating Curve= 0 ,0
Exp/Cntr(USF)=0,0
Exp/Cntr=0.3,0.1

Type RM Length L Ch R = 1 ,6987    ,328.7,329.9,327.8
XS GIS Cut Line= 2
2222383.62238928486066.9832077272221943.58878313485575.624079767
#Sta/Elev= 30
       0 3219.99    45.4 3208.17    85.9 3195.86    97.2 3189.47     117 3172.33
   125.5 3168.44   152.8 3167.77   174.2 3169.97   230.3 3171.01   249.4 3170.06
   255.8 3168.18   260.2 3167.11   278.5 3168.13     304 3169.63   340.8 3169.06
   366.3 3169.99   378.3 3169.09     432 3171.38   442.7 3169.44   465.5 3169.16
   482.4 3165.99   490.9 3168.12   502.3 3167.77   524.9 3170.72   536.3 3178.24
   564.6 3203.09   580.8 3212.21   609.2 3226.63   632.6 3242.11   659.6 3262.01
#Mann= 4 ,-1,0
       0      .1       0   255.8    .045       0   278.5      .1       0
   580.8     .06       0
#XS Ineff= 2 ,-1
       0  227.68 3173.09     320   431.5 3173.09
Permanent Ineff=
       F       F
Bank Sta=255.8,278.5
XS Rating Curve= 0 ,0
Exp/Cntr=0.3,0.1

Type RM Length L Ch R = 1 ,6657    ,187.5,185.7,185.7
XS GIS Cut Line= 2
2222582.37824699485884.3043679482222184.95168631485404.266668248
#Sta/Elev= 30
       0 3215.95    66.4 3193.05   114.6 3179.99   128.7 3173.16   135.2 3166.76
   141.4 3163.14   159.8 3164.12   172.8 3162.19   185.6 3163.76   210.4 3161.93
   233.9 3162.66   248.1 3159.47   258.5 3161.76   268.9 3161.21   293.73161.275
   310.4 3162.33   327.7 3160.09   336.4 3160.73   346.8 3164.74   367.6 3163.35
   404.4 3165.21   429.9 3161.97   445.5 3164.27   489.8 3163.19     513 3161.26
   518.2 3163.25     535 3177.38     572 3203.08   586.2 3210.67   623.2 3221.45
#Mann= 4 ,-1,0
       0      .1       0   268.9    .045       0   293.7      .1       0
     572     .06       0
#XS Ineff= 2 , 0
           216.7    3165
Permanent Ineff=
       F       F
Bank Sta=268.9,293.7
XS Rating Curve= 0 ,0
Exp/Cntr(USF)=0,0
Exp/Cntr=0.3,0.1

Type RM Length L Ch R = 1 ,6471    ,337.6,339.4,342.3
XS GIS Cut Line= 2
2222717.71466511 485781.694119312222288.07796549485217.602769082
#Sta/Elev= 30
       0 3216.63    91.2 3184.14   107.1 3179.69   127.1 3170.31   136.4 3164.89
     147  3160.6   156.5 3159.51   218.4 3158.79   231.9 3157.05   252.6  3155.9
   268.8 3156.99   297.3 3159.27   341.1 3158.77   365.6 3159.79   383.9 3158.67
     428  3158.7   443.9 3157.07   484.5 3165.03   510.9 3177.17   533.6 3192.63
   550.5 3197.54   563.7 3202.09   623.7 3218.45   629.7  3221.2   639.2 3222.53
   649.4 3225.45   680.8  3236.2   689.5 3240.76   697.9 3241.77   709.1  3241.4
#Mann= 5 ,-1,0
       0      .1       0   231.9    .045       0   268.8      .1       0
   550.5     .06       0   709.1      .1       0
#XS Ineff= 2 ,-1
       0   204.1    3163   297.3     413    3163
Permanent Ineff=
       F       F
Bank Sta=231.9,268.8
XS Rating Curve= 0 ,0
Exp/Cntr(USF)=0,0
Exp/Cntr=0.3,0.1

Type RM Length L Ch R = 1 ,6132    ,298.1,297.2,297.6
XS GIS Cut Line= 3
2222918.62391314485656.512203232 2222808.8965546485367.511977225
2222672.89644825485120.239056577
#Sta/Elev= 30
       0 3227.27    29.2 3214.86    89.1 3187.46   106.3 3176.84   134.7 3157.33
   140.5 3154.54   157.6 3149.17   187.2  3151.5   200.4 3149.32   208.9 3151.31
   230.3 3151.91   252.6 3151.65   264.6 3149.44   273.1 3150.67   325.5 3150.79
   333.5 3149.24   339.2 3148.21   348.3 3148.02   364.4 3149.13   371.1 3150.37
   407.7 3150.75   416.8 3153.36   425.9 3154.84     435 3159.25   448.7 3169.98
   457.9  3173.7   511.7 3186.92   526.4 3191.54   570.6 3202.73   591.3 3208.39
#Mann= 4 ,-1,0
       0      .1       0   333.5    .045       0   364.4      .1       0
   570.6     .06       0
Bank Sta=333.5,364.4
XS Rating Curve= 0 ,0
Exp/Cntr(USF)=0,0
Exp/Cntr=0.3,0.1

Type RM Length L Ch R = 1 ,5835    ,263.2,260,260.3
XS GIS Cut Line= 2
2223210.71505066 485480.330247272222901.62389985484948.693467877
#Sta/Elev= 30
       0 3216.53    26.8 3204.41   109.5 3174.73   123.3 3165.58   137.8 3152.63
   150.5 3146.84   167.5 3144.42   197.3 3142.69   230.4 3146.54   249.9 3144.18
   281.3 3143.46   300.1 3142.81     309 3143.47   314.3 3144.43   337.7 3144.62
   346.5 3142.89   358.2 3142.42   375.7 3145.52   384.5 3145.26   401.6 3147.51
   416.7 3154.59   433.9 3161.21   460.6 3167.26   472.3 3168.97   501.6 3176.61
   530.3 3183.27   572.8 3196.69   591.3 3203.84   600.5 3205.91     615 3213.63
#Mann= 4 ,-1,0
       0      .1       0   281.3    .045       0     309      .1       0
   501.6     .06       0
Bank Sta=281.3,309
XS Rating Curve= 0 ,0
Exp/Cntr(USF)=0,0
Exp/Cntr=0.3,0.1

Type RM Length L Ch R = 1 ,5575    ,246.1,251.9,262.6
XS GIS Cut Line= 3
2223404.55991053485443.0878495812223341.26191618  485234.1039952
 2223158.4010436484901.538342315
#Sta/Elev= 30
       0 3224.83    10.4 3219.42    52.1 3203.22    89.8 3186.49   131.6 3169.68
   160.8 3154.98   185.9 3138.73   198.4 3137.56   233.1 3140.55   237.7 3138.84
   242.2 3135.35   245.5 3135.03   260.5 3137.71   287.9 3138.89     297 3137.25
   315.3 3139.59   328.8 3139.91   342.7 3138.81     402 3139.81   420.8 3138.46
   437.8 3138.66   443.1 3140.53   453.1 3140.15   461.4 3142.22   484.2 3155.19
   496.7 3160.44   516.1 3165.67   548.1 3171.09     580 3179.95   597.9 3183.62
#Mann= 3 ,0,0
       0      .1       0   420.8    .045       0   437.8      .1       0
Bank Sta=420.8,437.8
XS Rating Curve= 0 ,0
Exp/Cntr(USF)=0,0
Exp/Cntr=0.3,0.1

Type RM Length L Ch R = 1 ,5323    ,217.3,205.9,202.4
XS GIS Cut Line= 3
  2223545.344824485407.1792959172223483.11856934485100.697894091
2223513.47921423484845.671662961
#Sta/Elev= 30
       0 3214.36    14.3 3208.81      51 3191.93   104.1 3171.01   128.6  3158.4
   153.1 3142.99   165.3 3137.76   173.5 3136.19   206.1 3134.08   234.7 3134.36
     247 3133.18   259.2 3130.47   263.3 3130.61   271.4 3133.31   287.8 3133.01
   308.2 3136.15   332.4 3135.41  346.95 3133.36   365.8  3133.3   381.6  3135.5
     421 3134.76   433.1  3136.6   441.2 3135.01   465.3 3134.81   477.4 3140.75
   489.6 3148.87   517.7 3163.96   525.7 3169.16   537.8  3174.6   569.6 3185.78
#Mann= 4 ,-1,0
       0      .1       0  346.95    .045       0   365.8      .1       0
  610.37     .06       0
#XS Ineff= 2 , 0
                          394.15         3138.99
Permanent Ineff=
       F       F
Bank Sta=346.95,365.8
XS Rating Curve= 0 ,0
Exp/Cntr(USF)=0,0
Exp/Cntr=0.3,0.1

Type RM Length L Ch R = 1 ,5117    ,211.5,211.7,212.4
XS GIS Cut Line= 2
2223694.74223372485418.2818532062223600.46943272484824.826843651
#Sta/Elev= 30
       0 3221.39    17.5 3212.41    29.5 3208.05   106.4 3176.41     151 3161.34
   195.7  3149.7   203.6 3146.11   223.9 3133.15   237.4 3128.52   254.8 3127.49
   265.3 3128.39   272.5 3130.28   304.9 3130.86     313 3131.68   333.2 3131.95
   345.4 3130.85   365.6 3132.74   377.8 3132.79   418.3 3131.92   434.5 3134.68
   446.6 3133.44   458.8 3134.47   466.9 3133.17     479  3132.5   483.1  3133.8
   499.3 3142.12   543.8 3166.43   564.1 3172.98   588.4 3181.94   600.9 3185.56
#Mann= 4 ,-1,0
       0      .1       0   237.4    .045       0   265.3      .1       0
     570     .06       0
#XS Ineff= 2 , 0
                          376.82         3134.73
Permanent Ineff=
       F       F
Bank Sta=237.4,265.3
XS Rating Curve= 0 ,0
Exp/Cntr(USF)=0,0
Exp/Cntr=0.3,0.1

Type RM Length L Ch R = 1 ,4905    ,136,137.4,138.8
XS GIS Cut Line= 2
2223898.57099751485400.6948867482223818.63902994484794.665241743
#Sta/Elev= 30
       0  3221.3      52 3195.95    64.1 3191.53    84.2 3181.14    96.3 3177.87
   108.4 3171.82   136.7 3160.74   164.9 3152.19   209.3 3141.27   217.4  3138.3
   233.5 3128.88   237.6  3127.3   245.6 3125.92   253.7 3125.93   261.8 3123.75
   273.9 3122.58     286 3122.84  288.05  3123.8   294.1 3127.16   366.7 3126.45
   390.9 3126.81     403    3128   427.2 3127.57   435.3  3125.7   447.4 3128.13
   483.7 3130.25   507.8 3138.77   536.1 3150.46   582.7 3164.73   611.3  3175.2
#Mann= 3 ,-1,0
       0      .1       0   261.8    .045       0  288.05      .1       0
#XS Ineff= 2 , 0
                           306.1         3129.61
Permanent Ineff=
       F       F
Bank Sta=261.8,288.05
XS Rating Curve= 0 ,0
Exp/Cntr(USF)=0,0
Exp/Cntr=0.3,0.1

Type RM Length L Ch R = 1 ,4768    ,87.7,87.4,87.1
BEGIN DESCRIPTION:
xs 4
END DESCRIPTION:
XS GIS Cut Line= 2
2224013.44605384485396.3544025262223979.54748013484731.894862235
#Sta/Elev= 30
       0 3218.38     7.2 3216.09    71.3 3183.83   132.8 3159.02   159.4 3150.15
   196.2 3139.98   247.5 3124.11   263.5 3123.63  273.56  3121.7   279.5 3120.32
   291.6 3120.54  297.16  3121.7   303.6 3124.65   307.6 3125.48   363.6 3124.91
   387.7 3123.42   407.7 3123.82   427.7  3122.1   443.8 3122.33   455.8 3124.57
   467.8 3125.14   535.9 3123.64   539.9 3124.73     553 3133.33   588.7 3152.22
     604 3161.88     640 3176.42     652 3182.68     660 3187.98   665.3 3189.54
#Mann= 4 ,-1,0
       0      .1       0  273.56    .045       0  297.16      .1       0
     640     .06       0
#XS Ineff= 2 , 0
                           307.6         3127.66
Permanent Ineff=
       F       F
Bank Sta=273.56,297.16
XS Rating Curve= 0 ,0
Exp/Cntr=0.5,0.3

Type RM Length L Ch R = 1 ,4681    ,41.6,40.4,41
BEGIN DESCRIPTION:
xs 3
END DESCRIPTION:
XS GIS Cut Line= 3
2224093.16122661485392.0628791852224089.40576913485154.217238637
2224060.61392843 484758.64238383
#Sta/Elev= 30
       0 3201.83    74.9 3173.53    98.9 3166.61   126.9 3156.27   138.9 3154.48
   158.9 3146.95   206.9 3134.22   222.9 3128.98   251.2 3126.97     259 3124.75
   269.6  3119.9     279 3118.71   292.3 3119.73   299.1 3123.19   303.1 3123.83
   355.9 3122.66   399.3 3124.09   407.4 3123.69   423.4 3120.97   439.4 3122.43
   455.5 3121.65   467.5 3119.91   475.5 3122.31   531.7 3122.87   539.7 3125.08
   555.8 3133.12   567.8 3140.87   595.2 3152.62   607.9  3161.4   634.5  3169.9
#Mann= 3 ,0,0
       0      .1       0   269.6    .045       0   292.3      .1       0
#XS Ineff= 3 ,-1
       0   259.6  3126.3   302.3     320 3121.86     320  590.04 3125.75
Permanent Ineff=
       F       F       F
Bank Sta=269.6,292.3
XS Rating Curve= 0 ,0
Exp/Cntr(USF)=0,0
Exp/Cntr=0.5,0.3

Type RM Length L Ch R = 1 ,4640    ,109.1,110.2,111.2
BEGIN DESCRIPTION:
xs 2
END DESCRIPTION:
XS GIS Cut Line= 3
2224130.71580143485392.0628791852224129.46398227485146.706323672
2224098.16850325484753.635107187
#Sta/Elev= 30
       0 3201.13    92.8 3167.58   126.9 3157.34   138.9 3154.54   154.9 3148.55
   198.9 3137.96   206.9 3134.54   210.9 3131.29   214.9 3130.04   246.9 3127.33
   262.8 3119.39     275 3118.28     287 3119.58     295 3122.57   299.1 3122.94
   375.3  3122.2   411.4 3123.59   427.5 3122.98   435.5 3119.94   451.5 3120.63
   459.6 3119.25   479.6 3121.44   499.7 3120.84   507.2 3122.54   527.8 3130.42
   535.8  3134.4   543.8 3136.95   551.9 3142.08   563.9  3147.1   639.7  3168.5
#Mann= 4 ,-1,0
       0      .1       0   262.8    .045       0     287      .1       0
   639.7     .06       0
#XS Ineff= 3 ,-1
       0   255.6    3126     294     305 3121.06     305  575.66 3125.41
Permanent Ineff=
       F       F       F
Bank Sta=262.8,287
XS Rating Curve= 0 ,0
Exp/Cntr(USF)=0,0
Exp/Cntr=0.5,0.3

Type RM Length L Ch R = 1 ,4530    ,120.3,119.1,118.9
BEGIN DESCRIPTION:
xs 1
END DESCRIPTION:
XS GIS Cut Line= 2
2224241.85965767485398.0348667212224231.03030676484767.968358735
#Sta/Elev= 30
       0 3209.87    12.9 3202.46    20.9 3199.68    68.9 3178.17    80.9 3174.05
   117.2 3159.38   140.9 3151.32   164.9 3143.71   178.3 3140.96   188.9 3136.67
   208.9 3135.83   224.9 3130.32   244.9 3125.34   256.9 3121.24   277.8 3117.75
   292.9 3116.64   301.4 3117.75   316.9 3121.26   341.1 3121.68   380.9 3119.16
   396.9 3119.81   427.3 3119.15   472.9 3120.34   476.9 3119.88   484.9 3117.16
   516.9 3117.48   521.7 3119.36   532.9  3126.2   552.9 3135.91   630.2 3154.76
#Mann= 3 ,-1,0
       0      .1       0   277.8    .045       0   301.4      .1       0
#XS Ineff= 2 , 0
                           340.4            3125
Permanent Ineff=
       F       F
Bank Sta=277.8,301.4
XS Rating Curve= 0 ,0
Exp/Cntr=0.3,0.1

Type RM Length L Ch R = 1 ,4411    ,83.2,78.7,74.6
BEGIN DESCRIPTION:
xs 4
END DESCRIPTION:
XS GIS Cut Line= 2
2224366.13590247485374.2255919952224342.02238081484775.406470787
#Sta/Elev= 30
       0 3197.91    13.1 3191.27    53.1 3175.38    68.3 3168.06   129.2 3144.59
   141.2 3140.87   149.2 3136.19   153.2 3135.23   169.2 3134.45   185.2 3129.22
   201.2 3126.39   213.2  3125.3   225.2 3122.69   241.5  3116.3   249.2    3115
   265.3 3115.18   269.3 3116.27   277.3 3119.02   305.3 3119.43   413.4 3117.74
   433.4 3116.29   457.4 3117.12   476.2 3114.52   485.4 3116.47   497.4 3114.11
   501.5 3114.01   505.5 3115.05   517.5 3122.67   541.3  3134.8   599.3 3149.63
#Mann= 3 ,-1,0
       0      .1       0   241.5    .045       0   269.3      .1       0
#XS Ineff= 2 , 0
                          303.21         3123.49
Permanent Ineff=
       F       F
Bank Sta=241.5,269.3
XS Rating Curve= 0 ,0
Exp/Cntr(USF)=0,0
Exp/Cntr=0.5,0.3

Type RM Length L Ch R = 1 ,4332    ,22.5,21.9,21.9
BEGIN DESCRIPTION:
xs 3
END DESCRIPTION:
XS GIS Cut Line= 6
2224457.73515146 485367.562456882224446.40839893  485151.0956306
2224428.15974206485092.574075821 2224420.6085737485078.730267163
2224404.24770892485059.2230822372224394.80874848484753.400763714
#Sta/Elev= 30
       0 3194.08    18.4 3184.52    46.4 3173.84    78.5 3159.95   134.5 3139.88
   174.6 3129.54   190.6 3123.91   214.7 3121.62   231.4 3121.06   235.6 3120.09
   246.8 3114.75     252 3113.16   256.5 3112.94   264.9 3113.17     268 3114.74
   273.3 3117.81   277.5 3118.25   329.4 3118.34   365.4 3118.71   393.4 3116.12
   429.4 3116.38   445.4 3116.12   457.4 3113.54   465.4 3113.21   490.7 3113.88
   505.5 3117.52   521.5 3127.33   540.2 3135.09   597.5 3146.21   625.3 3153.61
#Mann= 5 ,-1,0
       0      .1       0   246.8    .045       0     268      .1       0
   329.4     .07       0   429.4      .1       0
#XS Ineff= 3 ,-1
       0   242.6 3120.44     272     336 3118.33     336     600 3121.08
Permanent Ineff=
       F       F       F
Bank Sta=246.8,268
XS Rating Curve= 0 ,0
Exp/Cntr(USF)=0,0
Exp/Cntr=0.5,0.3

Type RM Length L Ch R = 1 ,4310    ,113.8,117.8,121.3
BEGIN DESCRIPTION:
xs 2
END DESCRIPTION:
XS GIS Cut Line= 6
2224479.13012848 485365.045400762224469.69116803485154.241950749
2224447.66692699485083.1351153732224438.22796654485066.774250596
2224421.86710176485049.7841217892224412.42814131484769.132364461
#Sta/Elev= 30
       0 3192.77    75.9 3159.05      84 3157.38   103.9 3148.95   119.9 3143.29
   168.9 3129.22     188 3122.79   208.1 3120.65   237.3 3119.95   243.83114.256
   245.7 3113.01   249.9 3112.73   262.4 3112.81   267.5  3114.2   270.8 3117.48
     275 3118.24   324.6 3118.51   372.4 3118.25   392.6 3115.32   428.6 3115.82
   444.6 3115.91   452.6 3112.62   472.7 3113.04   488.7 3115.83   504.4 3116.89
   512.2 3119.57   524.7 3126.54   544.7 3132.39   568.7 3141.09   608.8 3148.85
#Mann= 5 ,-1,0
       0      .1       0   243.8    .045       0   267.5      .1       0
   324.6     .07       0   428.6      .1       0
#XS Ineff= 3 ,-1
       0  240.28  3118.5  269.47     360  3116.9     360   560.3 3119.06
Permanent Ineff=
       F       F       F
Bank Sta=243.8,267.5
XS Rating Curve= 0 ,0
Exp/Cntr(USF)=0,0
Exp/Cntr=0.5,0.3

Type RM Length L Ch R = 1 ,4192    ,149,148.8,147.6
XS GIS Cut Line= 3
2224596.98886204485412.3301940922224558.35246819484900.784339501
2224535.17063188484698.329635721
#Sta/Elev= 30
       0 3196.75    31.2 3183.12    39.3 3181.24    71.4 3168.32    87.4 3160.71
   103.4 3150.66   115.5 3150.12   131.5 3143.21   143.6 3139.69   151.6 3135.31
   180.4 3131.36   207.7 3123.52   243.8 3117.32     292 3116.69     304 3111.08
   325.3  3111.1   336.1 3115.11   400.3 3113.23   452.4 3113.54   480.5 3110.11
   492.6 3110.79   500.6 3113.87   508.6 3114.32   565.2 3112.93   597.2 3114.95
   601.2 3116.35   630.2 3135.75   661.6 3145.82   673.7  3151.8   716.8  3164.9
#Mann= 3 ,0,0
       0      .1       0     304    .045       0   325.3      .1       0
#XS Ineff= 2 , 0
                          406.32         3116.24
Permanent Ineff=
       F       F
Bank Sta=304,325.3
XS Rating Curve= 0 ,0
Exp/Cntr(USF)=0,0
Exp/Cntr=0.3,0.1

Type RM Length L Ch R = 1 ,4044    ,190.8,178.2,165.5
XS GIS Cut Line= 3
2224870.99996955485336.953071578 2224735.9333759485192.238864089
2224665.64361797484718.127555744
#Sta/Elev= 30
       0 3144.79    21.6 3140.91    33.5 3141.72    48.9 3138.87    81.8 3135.87
    98.2 3133.05   112.2 3128.85   158.4 3122.97   261.7 3116.69   306.2 3115.79
   316.6 3109.71   344.8 3109.54   350.7 3113.11   370.9 3113.34   446.9  3110.8
   463.9  3106.7   488.1 3110.67   512.4 3108.38   524.5  3111.2   540.7 3110.93
   552.8 3108.36     565 3111.35   580.8 3110.74   589.2 3108.94   601.4 3110.77
   619.7  3115.6   637.8 3124.56     662 3146.49   670.1 3152.68   677.2 3156.15
#Mann= 4 ,-1,0
       0      .1       0   316.6    .045       0   344.8      .1       0
  637.95     .06       0
#XS Ineff= 2 , 0
                          408.56         3117.49
Permanent Ineff=
       F       F
Bank Sta=316.6,344.8
XS Rating Curve= 0 ,0
Exp/Cntr(USF)=0,0
Exp/Cntr=0.3,0.1

Type RM Length L Ch R = 1 ,3866    ,261.6,284.1,294.7
XS GIS Cut Line= 4
2224998.80735809485373.6938002412224909.17092436485022.875344071
2224836.53450392484956.4207466472224805.62538884484689.056901196
#Sta/Elev= 30
       0 3166.73    50.1 3155.97    62.5 3150.26    87.2 3151.19    99.6 3146.54
   157.4 3133.14   190.4 3115.55   202.8 3110.54   215.2 3108.59     230 3108.92
   351.5 3111.34   382.4 3110.66   388.3 3107.66     415 3107.48   447.6 3108.99
   455.6 3112.18   495.7 3111.76   516.1 3107.58   556.4  3103.7   564.5  3104.6
   576.5 3109.05   592.7 3109.58   612.8 3107.14   636.8 3110.97   651.5 3118.14
   681.2 3140.58   701.4 3152.29   713.5 3156.52   721.5 3161.56   729.7 3162.78
#Mann= 6 ,-1,0
       0      .1       0     230     .05       0     340      .1       0
   388.3    .045       0     415      .1       0  670.54     .06       0
#XS Ineff= 2 , 0
          297.46 3113.45  491.72         3114.16
Permanent Ineff=
       F       F
Bank Sta=388.3,415
XS Rating Curve= 0 ,0
Exp/Cntr(USF)=0,0
Exp/Cntr=0.3,0.1

Type RM Length L Ch R = 1 ,3581    ,151.1,146.5,142.8
XS GIS Cut Line= 3
2225088.03323421485339.1814613532224987.75494763485003.467197573
2224997.92810713484679.379401803
#Sta/Elev= 30
       0 3170.98    10.4  3167.9    18.8 3162.09    39.7 3160.76    52.2 3154.38
    98.1 3144.61   117.2 3139.12   126.9 3134.96   164.9 3112.25   171.9 3110.24
   185.8 3109.39   200.8 3106.18     283 3109.79   372.7 3109.75   472.7 3106.38
   516.7 3103.27   534.1 3104.56   540.8 3104.06     547 3101.84   556.8 3100.39
   574.2  3101.7   584.8  3108.7   592.8 3117.99   596.8 3121.35   616.8 3134.62
   644.8 3144.31   652.8 3148.74   660.8 3150.08   668.8 3154.28   674.6 3155.41
#Mann= 5 ,-1,0
       0      .1       0  400.37     .05       0  500.37      .1       0
     547    .045       0   574.2      .1       0
Bank Sta=547,574.2
XS Rating Curve= 0 ,0
Exp/Cntr(USF)=0,0
Exp/Cntr=0.3,0.1

Type RM Length L Ch R = 1 ,3435    ,142.1,135.9,130.6
XS GIS Cut Line= 3
2225279.94569436 485216.69049526 2225152.4346928484878.784848721
2225116.59906145484659.372652261
#Sta/Elev= 30
       0 3159.41    42.2 3147.14    59.3 3141.41    70.8 3134.67    76.4  3132.8
    93.5 3132.14   111.2 3128.85   135.3 3122.59   174.8  3110.2   198.1 3106.35
   225.9  3103.5   366.3 3104.82   411.2 3104.35   415.5  3103.2   420.9 3099.95
   423.6 3098.83   431.7 3098.48   447.9 3098.64   453.4 3099.78   460.1 3101.74
   476.3  3102.3   488.4 3104.32   498.7 3110.47   508.7 3120.91   512.6 3124.12
   526.5 3126.31   557.3  3137.3   565.4 3141.21   577.6 3149.43   583.5 3150.26
#Mann= 6 ,-1,0
       0      .1       0     290     .05       0  401.16     .06       0
   420.9    .045       0   453.4     .06       0  491.16      .1       0
Bank Sta=420.9,453.4
XS Rating Curve= 0 ,0
Exp/Cntr(USF)=0,0
Exp/Cntr=0.3,0.1

Type RM Length L Ch R = 1 ,3299    ,116,115.4,114.6
XS GIS Cut Line= 2
2225429.07012811485105.8703360842225213.03732834484643.660624958
#Sta/Elev= 30
       0 3137.64     9.6 3134.99    52.3 3119.13    71.4  3107.1    80.2 3102.41
    93.5 3099.89     106 3100.83   115.5 3100.19   190.8 3100.19   217.1 3101.46
   278.9 3102.33     295 3100.86   326.2 3099.73   349.6 3100.53   367.2 3100.27
   371.3 3099.82  375.453098.024   380.3 3096.76   392.4 3096.68   404.4 3096.82
   411.73097.939   424.6 3101.05   433.5  3102.2   437.9 3104.79   446.7  3111.8
   464.4  3120.5   473.2 3125.63   499.7 3143.89   504.1 3145.88   510.2 3146.66
#Mann= 8 ,-1,0
       0      .1       0      60     .06       0     170     .07       0
     210     .05       0     280      .1       0  375.45    .045       0
   411.7      .1       0     500     .06       0
#XS Ineff= 2 , 0
          277.14 3103.78
Permanent Ineff=
       F       F
Bank Sta=375.45,411.7
XS Rating Curve= 0 ,0
Exp/Cntr(USF)=0,0
Exp/Cntr=0.3,0.1

Type RM Length L Ch R = 1 ,3184    ,120.3,120.1,119.9
XS GIS Cut Line= 2
2225545.61010713485065.3135482362225321.33410385484609.584709584
#Sta/Elev= 30
       0 3138.22    22.4 3130.83    35.8 3127.22    49.2 3121.63    58.1 3118.71
    69.9 3112.46    80.4 3107.91    84.9 3105.31    87.8 3103.13    98.2 3097.49
   102.5  3096.9   116.1 3096.99   129.6 3098.25   182.9 3098.05   200.8 3098.98
   223.1 3099.45   317.9 3099.36   330.1 3098.31   396.9 3096.75  400.87 3095.62
   405.8 3094.69   419.2 3094.53   428.1 3094.68   431.4 3095.67     437 3097.81
   446.4 3099.77   476.2 3122.24   481.6 3125.27   486.1 3127.11   507.9 3140.68
#Mann= 7 ,-1,0
       0      .1       0      20     .05       0     130     .06       0
     240      .1       0  400.87    .045       0   431.4      .1       0
     460     .06       0
#XS Ineff= 2 , 0
          239.64 3101.24
Permanent Ineff=
       F       F
Bank Sta=400.87,431.4
XS Rating Curve= 0 ,0
Exp/Cntr(USF)=0,0
Exp/Cntr=0.3,0.1
